--- MEADOWCK1.prj (project) ---

Proj Title=MEADOWCK1
Current Plan=p01
Default Exp/Contr=0.3,0.1
English Units
Geom File=g01
Flow File=f01
Plan File=p01
Y Axis Title=Elevation
X Axis Title(PF)=Main Channel Distance
X Axis Title(XS)=Station
BEGIN DESCRIPTION:
Stream Name- Meadow Creek 1
Flood Zone: Zone A
Greenbrier County, WV
County-Wide Study
WVDHSEM-2018-3, Flood Risk Project
HEC-RAS Version: 5.0.7
General Notes:
For the Hydrology Regression was used.
END DESCRIPTION:
DSS Export Rating Curves= 0
DSS Export Rating Curve Sorted= 0
DSS Export Volume Flow Curves= 0
DXF Filename=A2c.
DXF OffsetX= 0
DXF OffsetY= 0
DXF ScaleX= 1
DXF ScaleY= 10

--- MEADOWCK1.p01 (plan) ---

Plan Title=Floodplain
Program Version=5.07
Short Identifier=Floodplain
Geom File=g01
Flow File=f01
Subcritical Flow
K Sum by GR= 0
Std Step Tol= 0.01
Critical Tol= 0.01
Num of Std Step Trials= 20
Max Error Tol= 0.3
Flow Tol Ratio= 0.001
Split Flow NTrial= 30
Split Flow Tol= 0.02
Split Flow Ratio= 0.02
Log Output Level= 0
Friction Slope Method= 1
Unsteady Friction Slope Method= 2
Unsteady Bridges Friction Slope Method= 1
Parabolic Critical Depth
Global Vel Dist= 0 , 0 , 0
Global Log Level= 0
CheckData=True
Encroach Param=-1 ,0,0, 0
Computation Interval=1MIN
Output Interval=1HOUR
Instantaneous Interval=1HOUR
Mapping Interval=1HOUR
Computation Time Step Use Courant=        0
Computation Time Step Use Time Series=    0
Computation Time Step Count To Double=0
Computation Time Step Max Doubling=0
Computation Time Step Max Halving=0
Computation Time Step Residence Courant=0
Run HTab= 0
Run UNet= 0
Run Sediment= 0
Run PostProcess= 0
Run WQNet= 0
Run RASMapper= 0
UNET Theta= 1
UNET Theta Warmup= 1
UNET ZTol= 0.02
UNET ZSATol= 0.02
UNET MxIter= 20
UNET Max Iter WO Improvement= 0
UNET MaxInSteps= 0
UNET DtIC= 0
UNET DtMin= 0
UNET MaxCRTS= 20
UNET WFStab= 2
UNET SFStab= 1
UNET WFX= 1
UNET SFX= 1
UNET 1D Methodology=Finite Difference
UNET DSS MLevel= 4
UNET Pardiso=0
UNET DZMax Abort= 100
UNET Use Existing IB Tables=-1
UNET Froude Reduction=False
UNET Froude Limit= 0.8
UNET Froude Power= 4
UNET D1 Cores= 0
UNET D2 Coriolis=0
UNET D2 Cores= 0
UNET D2 Theta= 1
UNET D2 Theta Warmup= 1
UNET D2 Z Tol= 0.01
UNET D2 Volume Tol= 0.01
UNET D2 Max Iterations= 20
UNET D2 Equation= 0
UNET D2 RampUpFraction=0.1
UNET D2 TimeSlices= 1
UNET D2 BCVolumeCheck=0
UNET D1D2 MaxIter= 0
UNET D1D2 ZTol=0.01
UNET D1D2 QTol=0.1
UNET D1D2 MinQTol=1
Write IC File= 0
Write IC File at Fixed DateTime=0
Write IC File at Sim End=0
Echo Input=False
Echo Parameters=False
Echo Output=False
Write Detailed= 0
HDF Write Warmup=0
HDF Write Time Slices=0
HDF Flush=0
HDF Face Node Velocities=0
HDF Compression= 1
HDF Chunk Size= 1
HDF Spatial Parts= 1
HDF Use Max Rows=0
HDF Fixed Rows= 1
Calibration Method= 0
Calibration Iterations= 20
Calibration Max Change=0.05
Calibration Tolerance=0.2
Calibration Maximum=1.5
Calibration Minimum=0.5
Calibration Optimization Method= 1
WQ AD Non Conservative
WQ ULTIMATE=-1
WQ Max Comp Step=1HOUR
WQ Output Interval=15MIN
WQ Output Selected Increments= 0
WQ Output face flow=0
WQ Output face velocity=0
WQ Output face area=0
WQ Output face dispersion=0
WQ Output cell volume=0
WQ Output cell surface area=0
WQ Output cell continuity=0
WQ Output cumulative cell continuity=0
WQ Output face conc=0
WQ Output face dconc_dx=0
WQ Output face courant=0
WQ Output face peclet=0
WQ Output face adv mass=0
WQ Output face disp mass=0
WQ Output cell mass=0
WQ Output cell source sink temp=0
WQ Output nsm pathways=0
WQ Output nsm derived pathways=0
WQ Output MaxMinRange=-1
WQ Daily Max Min Mean=-1
WQ Daily Range=0
WQ Daily Time=0
WQ Create Restart=0
WQ Fixed Restart=0
WQ System Summary=0
WQ Write To DSS=0
WQ Use Fixed Temperature=0
Sorting and Armoring Iterations= 10
XS Update Threshold= 0.02
Bed Roughness Predictor= 0
Hydraulics Update Threshold= 0.02
Energy Slope Method= 1
Volume Change Method= 1
Sediment Retention Method= 0
XS Weighting Method= 0
Number of US Weighted Cross Sections= 1
Number of DS Weighted Cross Sections= 1
Upstream XS Weight=0
Main XS Weight=1
Downstream XS Weight=0
Number of DS XS's Weighted with US Boundary= 1
Upstream Boundary Weight= 1
Weight of XSs Associated with US Boundary= 0
Number of US XS's Weighted with DS Boundary= 1
Downstream Boundary Weight= 0.5
Weight of XSs Associated with DS Boundary= 0.5
Percentile Method= 0
Sediment Output Level= 3
Mass or Volume Output= 0
Output Increment Type= 1
Profile and TS Output Increment= 1
XS Output Flag= 0
XS Output Increment= 10
Write Gradation File= 0
Read Gradation Hotstart= 0
Write HDF5 File= 1
Write Binary Output= 1
Write DSS Sediment File= 0
SV Curve= 0
Specific Gage Flag= 0

--- MEADOWCK1.f01 (steady flow) ---

Flow Title=Flow
Program Version=5.07
Number of Profiles= 6
Profile Names=f1p,f10p,f4p,f2p,f02p,f1pplus
River Rch & RM=MEADOWCK1,Main            ,75581
     529     279     371     448     740     782
River Rch & RM=MEADOWCK1,Main            ,73978
     598     316     420     506     834     884
River Rch & RM=MEADOWCK1,Main            ,71430
     678     361     478     575     945    1000
River Rch & RM=MEADOWCK1,Main            ,69203
     792     424     560     672    1100    1170
River Rch & RM=MEADOWCK1,Main            ,67339
     882     474     625     749    1220    1300
River Rch & RM=MEADOWCK1,Main            ,64109
    1010     548     721     863    1400    1500
River Rch & RM=MEADOWCK1,Main            ,61239
    1140     619     812     971    1570    1690
River Rch & RM=MEADOWCK1,Main            ,59576
    1280     700     917    1090    1770    1900
River Rch & RM=MEADOWCK1,Main            ,56054
    1450     794    1040    1240    1990    2140
River Rch & RM=MEADOWCK1,Main            ,50980
    1720     950    1240    1470    2360    2550
River Rch & RM=MEADOWCK1,Main            ,44209
    1940    1080    1400    1660    2650    2870
River Rch & RM=MEADOWCK1,Main            ,38864
    2190    1220    1580    1870    2980    3230
River Rch & RM=MEADOWCK1,Main            ,31946
    2500    1400    1810    2140    3390    3690
River Rch & RM=MEADOWCK1,Main            ,24140
    2780    1560    2020    2390    3780    4120
River Rch & RM=MEADOWCK1,Main            ,14473
    3730    2120    2720    3210    5030    5510
Boundary for River Rch & Prof#=LAURELRN2,Main            , 1
Up Type= 0
Dn Type= 3
Dn Slope=0.035124
Boundary for River Rch & Prof#=LAURELRN2,Main            , 2
Up Type= 0
Dn Type= 3
Dn Slope=0.035124
Boundary for River Rch & Prof#=LAURELRN2,Main            , 3
Up Type= 0
Dn Type= 3
Dn Slope=0.035124
Boundary for River Rch & Prof#=LAURELRN2,Main            , 4
Up Type= 0
Dn Type= 3
Dn Slope=0.035124
Boundary for River Rch & Prof#=LAURELRN2,Main            , 5
Up Type= 0
Dn Type= 3
Dn Slope=0.035124
Boundary for River Rch & Prof#=LAURELRN2,Main            , 6
Up Type= 0
Dn Type= 3
Dn Slope=0.035124
Boundary for River Rch & Prof#=MEADOWCK1,Main            , 1
Up Type= 0
Dn Type= 3
Dn Slope=0.011297
Boundary for River Rch & Prof#=MEADOWCK1,Main            , 2
Up Type= 0
Dn Type= 3
Dn Slope=0.011297
Boundary for River Rch & Prof#=MEADOWCK1,Main            , 3
Up Type= 0
Dn Type= 3
Dn Slope=0.011297
Boundary for River Rch & Prof#=MEADOWCK1,Main            , 4
Up Type= 0
Dn Type= 3
Dn Slope=0.011297
Boundary for River Rch & Prof#=MEADOWCK1,Main            , 5
Up Type= 0
Dn Type= 3
Dn Slope=0.011297
Boundary for River Rch & Prof#=MEADOWCK1,Main            , 6
Up Type= 0
Dn Type= 3
Dn Slope=0.011297
Boundary for River Rch & Prof#=MFANTNYCK,Main            , 1
Up Type= 0
Dn Type= 3
Dn Slope=0.001473
Boundary for River Rch & Prof#=MFANTNYCK,Main            , 2
Up Type= 0
Dn Type= 3
Dn Slope=0.001473
Boundary for River Rch & Prof#=MFANTNYCK,Main            , 3
Up Type= 0
Dn Type= 3
Dn Slope=0.001473
Boundary for River Rch & Prof#=MFANTNYCK,Main            , 4
Up Type= 0
Dn Type= 3
Dn Slope=0.001473
Boundary for River Rch & Prof#=MFANTNYCK,Main            , 5
Up Type= 0
Dn Type= 3
Dn Slope=0.001473
Boundary for River Rch & Prof#=MFANTNYCK,Main            , 6
Up Type= 0
Dn Type= 3
Dn Slope=0.001473
Boundary for River Rch & Prof#=NFANTNYCK,Main            , 1
Up Type= 0
Dn Type= 3
Dn Slope=0.006644
Boundary for River Rch & Prof#=NFANTNYCK,Main            , 2
Up Type= 0
Dn Type= 3
Dn Slope=0.006644
Boundary for River Rch & Prof#=NFANTNYCK,Main            , 3
Up Type= 0
Dn Type= 3
Dn Slope=0.006644
Boundary for River Rch & Prof#=NFANTNYCK,Main            , 4
Up Type= 0
Dn Type= 3
Dn Slope=0.006644
Boundary for River Rch & Prof#=NFANTNYCK,Main            , 5
Up Type= 0
Dn Type= 3
Dn Slope=0.006644
Boundary for River Rch & Prof#=NFANTNYCK,Main            , 6
Up Type= 0
Dn Type= 3
Dn Slope=0.006644
Boundary for River Rch & Prof#=TWOMILERN,Main            , 1
Up Type= 0
Dn Type= 3
Dn Slope=0.021324
Boundary for River Rch & Prof#=TWOMILERN,Main            , 2
Up Type= 0
Dn Type= 3
Dn Slope=0.021324
Boundary for River Rch & Prof#=TWOMILERN,Main            , 3
Up Type= 0
Dn Type= 3
Dn Slope=0.021324
Boundary for River Rch & Prof#=TWOMILERN,Main            , 4
Up Type= 0
Dn Type= 3
Dn Slope=0.021324
Boundary for River Rch & Prof#=TWOMILERN,Main            , 5
Up Type= 0
Dn Type= 3
Dn Slope=0.021324
Boundary for River Rch & Prof#=TWOMILERN,Main            , 6
Up Type= 0
Dn Type= 3
Dn Slope=0.021324
DSS Import GetInterval= 0
DSS Import GetPeak= 0
DSS Import FillOption= 0

--- MEADOWCK1.g01 (geometry) ---

Geom Title=Geometry
Program Version=5.07

River Reach=MEADOWCK1       ,Main
Reach XY= 30
2260734.90560606376864.4507299812258071.48540796374944.584819064
 2258373.9841468374052.8352902232257518.56722248373437.835207894
 2257496.7299958371967.9975963982256030.55018538371106.775237471
2255845.04104197 369043.663221972252537.49549171 364509.62209323
2250894.70842297360936.0675605542248280.36325797359114.362542555
2247574.76690014357540.1357041452246757.87319273357789.033500314
2244231.69222148355938.2734223162243774.74792539356245.217690304
2240513.63666546353574.3844493032239533.08121188353789.662233979
2238187.24794555 351831.328880312235241.41459839350288.967791811
2234698.35892597348830.6344223922233659.15988889348449.135185391
2233903.91464873347378.5510404712232503.91449597346949.384575978
2230215.02570106 344536.189927312227978.91468772343616.745571971
2226997.20109998 344011.42785348 2227523.2426988345054.657066226
2224355.18702705347149.7959205662221503.79837289351014.379398733
2219966.94908439351223.2546371372218873.18224305353280.180313304

Type RM Length L Ch R = 1 ,75581   ,131.2,133.7,135.5
XS GIS Cut Line= 4
2261175.92211246376713.2617278992260854.58515672376806.768758729
 2260576.6687178 376929.685507642260292.24146514377076.109099314
#Sta/Elev= 30
       0 2934.32   102.2 2908.98   146.7 2899.98   156.9 2899.14     184 2894.82
   201.3 2890.17   221.8 2889.11   253.4 2885.76   292.5 2882.89   331.2 2877.63
   384.6 2873.26   404.5 2870.08   427.9 2869.35   452.32865.346   460.1  2863.7
   467.3 2863.46  483.412864.858   492.4  2867.2   499.6 2867.88   524.7 2866.76
     557 2866.74   582.1 2868.85   596.5 2867.64   610.6 2869.53   639.5 2879.49
     658 2884.95   757.7 2909.13   827.7 2929.49   938.4 2956.66   958.5 2960.49
#Mann= 8 ,-1 , 0
       0      .1       0  301.28     .12       0  403.07     .06       0
   452.3    .045       0  483.41     .06       0  542.83      .1       0
  712.32      .1       0  784.42      .1       0
#XS Ineff= 2 , 0
                          498.24         2870.07
Permanent Ineff=
       F       F
Bank Sta=452.3,483.41
XS Rating Curve= 0 ,0
Exp/Cntr=0.3,0.1

Type RM Length L Ch R = 1 ,75447   ,144.1,143,145.3
XS GIS Cut Line= 2
2261036.21733938376613.4354839772260212.60612573 376906.49100022
#Sta/Elev= 30
       0 2932.96    44.6 2923.04    84.8 2916.58   133.5 2905.68   217.1  2892.1
   269.3 2879.62   311.1 2865.43     332 2862.76  348.042861.916   352.9 2860.76
   362.2 2860.27  365.852861.288   370.3 2862.79   377.3 2863.22   401.7    2861
   464.3 2862.26   471.3 2861.48   509.6 2863.09   523.5 2866.83   558.2 2878.57
   567.7 2880.51   637.9 2900.97   683.7 2918.49   696.9 2924.53   715.1 2930.92
   749.9 2945.68   781.2 2955.69   822.2 2966.31   840.4 2969.76   874.2 2973.62
#Mann= 8 ,-1 , 0
       0      .1       0  180.05     .12       0  281.02     .06       0
  348.04    .045       0  365.85     .06       0  406.73      .1       0
  583.95      .1       0   785.9      .1       0
#XS Ineff= 2 , 0
                          377.17         2864.69
Permanent Ineff=
       F       F
Bank Sta=348.04,365.85
XS Rating Curve= 0 ,0
Exp/Cntr=0.3,0.1

Type RM Length L Ch R = 1 ,75304   ,188.1,189.3,186.3
XS GIS Cut Line= 2
2260962.60626614376456.4909159842260177.88375422376824.546610311
#Sta/Elev= 30
       0 2941.41      25 2934.15   101.1 2915.86     170 2896.16   191.7 2891.54
   235.2  2883.8   246.1 2881.38   289.6  2870.6   312.7 2863.67   325.8 2861.44
   358.4 2858.24  372.832855.948   381.7 2854.83   402.32855.927   418.7 2857.41
   460.7 2856.62   474.4 2857.28   481.6 2857.93   521.5 2865.21   546.4 2872.63
   581.5 2887.54   612.1 2899.17   640.1 2910.98   666.4 2920.79   704.9 2936.69
   720.8 2942.77   742.5 2949.99   798.6 2965.59   829.5 2969.88   866.7 2972.43
#Mann= 6 ,-1 , 0
       0      .1       0  257.18     .06       0  372.83    .045       0
   402.3      .1       0  547.87      .1       0  754.44      .1       0
#XS Ineff= 2 , 0
                          448.22         2861.46
Permanent Ineff=
       F       F
Bank Sta=372.83,402.3
XS Rating Curve= 0 ,0
Exp/Cntr=0.3,0.1

Type RM Length L Ch R = 1 ,75115   ,155.7,155.2,153.3
XS GIS Cut Line= 2
2260877.88399464376306.4908878952260070.93941431 376684.26867564
#Sta/Elev= 30
       0  2941.4      22 2937.43    58.3 2928.68    72.7 2922.72   105.3 2913.55
     120 2907.82   181.4 2889.94   224.9 2874.31   257.5 2866.98   264.7 2864.45
   308.2 2857.34   358.9 2852.77   366.2 2852.91  379.472850.566   387.9 2849.29
  406.192849.981   420.5 2852.03   449.5 2851.55   470.4 2852.82   482.1 2854.65
   491.9 2857.67   532.1 2873.43   596.2 2906.84   648.7 2929.67   688.6 2944.06
     724 2953.34   752.7 2959.54   797.3 2963.78   815.4  2964.7     891 2965.18
#Mann= 7 ,-1 , 0
       0      .1       0  257.37     .06       0  379.47    .045       0
  406.19     .06       0  478.51      .1       0  485.79      .1       0
  692.32      .1       0
Bank Sta=379.47,406.19
XS Rating Curve= 0 ,0
Exp/Cntr=0.3,0.1

Type RM Length L Ch R = 1 ,74959   ,129.8,130.8,131
XS GIS Cut Line= 2
 2260779.2726433376155.1020830572259988.99502438376592.602192312
#Sta/Elev= 30
       0 2924.55    71.8 2904.09   115.2 2890.41   124.9 2888.77   145.4 2881.51
   206.3 2863.38   232.6 2858.05   266.3  2853.1   322.6 2849.38   351.8 2848.69
   371.1  2845.2  381.612844.726   392.8 2844.26  401.752845.287   438.7 2847.81
   455.6 2852.18     479  2863.8   517.6 2885.98   546.7 2900.59   570.1 2910.08
   611.3 2928.85   667.6  2947.3   690.1 2951.67   705.1 2953.47   742.8 2955.98
   765.1 2956.75   787.6 2956.16   806.3 2957.51   847.6 2956.86   903.3  2957.7
#Mann= 7 ,-1 , 0
       0      .1       0  223.87     .12       0  360.15     .06       0
  381.61    .045       0  401.75     .06       0  486.26      .1       0
  629.89      .1       0
Bank Sta=381.61,401.75
XS Rating Curve= 0 ,0
Exp/Cntr=0.3,0.1

Type RM Length L Ch R = 1 ,74829   ,161.8,161.7,161
XS GIS Cut Line= 3
 2260766.7726683376063.4352716512260413.99515864376212.046522975
2259988.01110247376417.601886138
#Sta/Elev= 30
       0 2915.82      15 2912.56    32.8 2907.07    59.8 2901.57    89.8 2894.27
   143.2  2878.2   242.8 2851.41   296.2 2847.07   321.2 2846.51   335.1 2845.31
   385.5 2844.42  411.962841.474   421.7 2840.29  432.072841.914   454.2 2841.62
   465.4 2843.11   483.7 2851.79   538.3 2880.85   549.2 2885.84   596.6 2902.72
   636.7 2920.29   653.2 2925.94   709.5 2939.37   738.7 2944.63   762.9 2946.17
   771.4    2946   796.9 2948.06   811.5 2947.52   818.8  2949.1   855.8 2948.98
#Mann= 7 ,-1 , 0
       0      .1       0  234.13     .12       0  382.24     .06       0
  411.96    .045       0  432.07     .06       0  504.38      .1       0
  615.58      .1       0
Bank Sta=411.96,432.07
XS Rating Curve= 0 ,0
Exp/Cntr=0.3,0.1

Type RM Length L Ch R = 1 ,74667   ,155.3,150.6,144.9
XS GIS Cut Line= 3
2260665.09439397 375896.421498062260134.57019256376179.812991649
2259941.48330839376318.643750727
#Sta/Elev= 30
       0 2903.54      38  2891.7    77.2 2882.08   129.2 2862.01   144.9  2858.9
   160.8 2857.99   205.4 2852.99   227.7 2852.15   254.5 2848.29   331.6 2841.97
   346.7 2840.17     368 2835.79   380.1 2836.82  398.662836.732   416.5 2835.17
  418.862835.994   424.9 2839.28   428.5 2840.02   447.2 2840.57   469.5 2842.95
   488.1 2847.08   506.7 2852.77   549.8 2868.94   614.9 2890.22     648 2903.97
     683 2915.78   700.5 2920.73     763  2934.4   801.6 2938.52   839.3 2940.35
#Mann= 6 ,-1 , 0
       0      .1       0  298.32     .12       0  336.81     .06       0
  398.66    .045       0  418.86     .06       0  533.29      .1       0
Bank Sta=398.66,418.86
XS Rating Curve= 0 ,0
Exp/Cntr=0.3,0.1

Type RM Length L Ch R = 1 ,74516   ,229.9,229.3,226.9
XS GIS Cut Line= 3
2260378.98341763375713.0882033112260115.09450972376128.365916058
2259934.53909655376311.699210808
#Sta/Elev= 30
       0 2906.56    24.6 2898.41    36.7 2893.58    71.7 2885.43    83.3 2880.59
   124.7 2866.87   145.5 2858.38   164.4 2849.62   179.3 2844.48   188.8 2842.38
     215 2838.87   246.6 2836.51   269.2    2836   283.9 2834.52   312.7 2834.07
  327.992832.288   339.9 2830.66  354.262832.496   363.2 2835.51   390.9 2837.39
   409.9 2841.77   471.7  2863.5   505.2 2876.92   553.4 2892.72   606.7 2914.87
   629.9 2921.91   647.9 2926.36   690.2 2934.04   728.5 2938.36   749.3 2939.13
#Mann= 5 ,-1 , 0
       0      .1       0  286.28     .06       0  327.99    .045       0
  354.26     .06       0  454.36      .1       0
Bank Sta=327.99,354.26
XS Rating Curve= 0 ,0
Exp/Cntr=0.3,0.1

Type RM Length L Ch R = 1 ,74287   ,312.5,308.9,301.6
XS GIS Cut Line= 2
2260135.92780139375631.1438133872259817.87233514376271.421404228
#Sta/Elev= 30
       0  2902.8    27.2 2894.77    51.1 2884.83    79.2 2869.69    96.3 2857.74
   111.4  2848.2   123.2 2842.26     148 2832.08   159.9 2830.29   195.7  2829.3
   221.3  2827.2     236 2826.83  250.572824.805   261.6 2823.39  275.472824.709
   294.5 2828.03     324 2827.47   349.5 2828.35   377.8 2831.54   400.8 2836.84
   412.5 2839.94   441.4 2849.45   473.2 2863.28   558.3 2895.85   569.3 2901.87
   609.6 2915.23   636.8 2923.33   653.6 2926.69   701.2 2934.21   714.9 2935.36
#Mann= 5 ,-1 , 0
       0      .1       0  246.66     .06       0  250.57    .045       0
  275.47     .06       0  364.51      .1       0
Bank Sta=250.57,275.47
XS Rating Curve= 0 ,0
Exp/Cntr=0.3,0.1

Type RM Length L Ch R = 1 ,73978   ,56.8,55.9,54.6
XS GIS Cut Line= 2
 2259741.4833803375590.8660068062259715.09465355376246.421454221
#Sta/Elev= 30
       0 2900.92    18.7 2897.44    35.1 2890.67    84.4 2876.77   117.2 2862.18
   149.6 2851.57   166.4 2842.98   176.3 2839.22   192.7 2830.35   209.1 2823.77
   222.2 2820.63   255.1 2817.16  262.482814.377   268.2 2812.92  282.532814.748
   301.1 2815.44   314.2 2818.99   342.1 2820.24   360.2 2822.71   372.9 2826.16
   383.2 2830.73   429.1 2856.18   445.5 2864.44   468.4 2874.76   504.6 2888.93
   544.1 2905.97   570.3 2914.07   603.1 2922.47   629.4 2927.74   656.1 2930.88
#Mann= 5 ,-1 , 0
       0      .1       0  164.51     .06       0  262.48    .045       0
  282.53     .06       0  297.28      .1       0
Bank Sta=262.48,282.53
XS Rating Curve= 0 ,0
Exp/Cntr=0.3,0.1

Type RM Length L Ch R = 1 ,73922   ,152.4,158.7,163.4
XS GIS Cut Line= 4
2259694.67817603375596.5903590752259666.78081495375767.461695682
2259684.21666562375961.3483551782259680.72949549376241.019399992
#Sta/Elev= 30
       0 2890.22    16.4 2886.14    56.3 2874.69    89.4 2861.84   131.1 2849.14
   151.4  2841.5   172.8 2832.68     185 2828.46   212.2 2820.75   230.3 2816.36
   238.6 2815.46   258.3  2816.3   272.42814.373   294.2 2814.38   297.9  2814.3
   301.2 2814.35   317.6 2817.13   350.6 2818.78   363.3 2822.56   373.6 2827.05
   396.6 2838.76   432.6  2858.9   455.6 2871.07   479.2 2880.32   508.1 2893.43
   526.6 2900.99   563.9 2913.59   593.4 2920.92   609.8 2924.11   647.5 2928.13
#Mann= 4 ,-1 , 0
       0      .1       0   151.4     .06       0   272.4    .045       0
   294.2      .1       0
Bank Sta=272.4,294.2
XS Rating Curve= 0 ,0
Exp/Cntr(USF)=0,0
Exp/Cntr=0.3,0.1

Type RM Length L Ch R = 1 ,73764   ,187,189,190.6
XS GIS Cut Line= 2
2259622.03906539375568.6436103142259399.81674081376199.199107721
#Sta/Elev= 30
       0 2881.34    14.8  2877.2    32.5 2873.61    60.7 2865.92    86.8 2855.64
   120.3 2846.64   140.9 2837.65   165.1 2830.88   221.1 2817.95   241.6 2814.03
   279.9 2811.28  285.122810.144   292.6 2809.11   307.7 2808.98   315.8 2810.15
   325.1 2811.93     339  2811.5     353 2812.88   373.8  2818.8   384.3 2822.63
   394.7 2827.04   412.1 2836.15   467.7 2868.06   492.1 2877.18   503.5 2885.08
   533.8 2898.21   552.4 2903.77   582.5 2910.18   644.5 2919.76   668.6 2922.23
#Mann= 6 ,-1 , 0
       0      .1       0  157.44     .06       0  284.45      .1       0
  285.12    .045       0   315.8      .1       0  571.56      .1       0
Bank Sta=285.12,315.8
XS Rating Curve= 0 ,0
Exp/Cntr=0.3,0.1

Type RM Length L Ch R = 1 ,73575   ,187.8,194,199.6
XS GIS Cut Line= 2
2259491.48355222 375532.532462062259170.65020439376096.421426147
#Sta/Elev= 30
       0 2860.44    13.1 2857.02    33.6 2850.11    69.7 2841.01   111.2 2825.12
   129.4 2820.08   152.8  2815.8   166.1 2814.72   192.4 2811.06   235.8 2807.99
   250.9 2805.86   273.6 2805.97  284.332803.753   298.3 2802.36  304.382803.634
   315.1 2806.22   329.5  2807.4   339.2 2810.11   360.4 2820.97   401.7 2847.27
   424.5 2860.34   439.6 2872.35   443.4 2874.52   467.7 2885.35   507.6 2898.01
   520.8  2901.8   550.9 2906.49   591.8 2909.25   632.1 2911.01   648.8    2911
#Mann= 5 ,-1 , 0
       0      .1       0   27.57     .12       0  166.94     .06       0
  284.33    .045       0  304.38      .1       0
Bank Sta=284.33,304.38
XS Rating Curve= 0 ,0
Exp/Cntr=0.3,0.1

Type RM Length L Ch R = 1 ,73381   ,280.2,274.9,270.9
XS GIS Cut Line= 3
2259455.37240396 375532.532462062259016.48351797375753.366009891
 2258898.4279798375843.643716484
#Sta/Elev= 30
       0  2851.1    41.5 2838.92    64.3 2829.84    69.1    2829    93.6 2820.92
   107.4 2817.68   139.2 2811.16   161.2 2807.67   189.1 2805.32   214.9 2801.21
   229.6 2800.49  239.552798.336   249.1 2796.27  259.56 2798.31   266.3 2798.35
   288.3 2802.17   299.3 2803.12   358.1 2805.41   376.2 2812.15   412.2 2830.95
   427.5 2839.99   449.9 2851.33   460.9 2858.15   486.1 2870.11   502.7 2875.59
   523.2 2880.96   556.6 2888.28   582.3 2891.59   618.2  2894.2   639.9 2894.98
#Mann= 6 ,-1 , 0
       0     .12       0    84.9      .1       0  224.25     .06       0
  239.55    .045       0  259.56     .06       0  350.79      .1       0
Bank Sta=239.55,259.56
XS Rating Curve= 0 ,0
Exp/Cntr=0.3,0.1

Type RM Length L Ch R = 1 ,73106   ,411.6,411.6,412.7
XS GIS Cut Line= 2
2259244.26127763375253.3660256422258806.76116839375792.254711643
#Sta/Elev= 30
       0 2826.65    15.7    2823    36.6 2820.03    73.7 2812.86   108.9 2804.46
   167.3  2796.2   172.6 2794.85   179.9 2791.11   184.1 2789.78   192.9 2789.28
   197.6 2789.63   202.2 2791.33   214.2 2793.95   253.6 2795.86   323.5 2795.22
   353.1 2792.84     370 2795.74   408.1 2794.25   428.5  2798.6   443.2 2803.81
   467.2 2809.67   498.5 2819.66   531.1 2834.15     589 2862.91   598.7 2867.25
   612.7 2872.08   627.8 2876.05   646.2 2879.54   674.3 2883.19   694.1 2883.71
#Mann= 7 ,-1 , 0
       0      .1       0  155.32     .12       0   179.9    .045       0
   202.2     .12       0  226.78      .1       0  288.38     .06       0
  433.78      .1       0
#XS Ineff= 2 , 0
                          244.03         2800.95
Permanent Ineff=
       F       F
Bank Sta=179.9,202.2
XS Rating Curve= 0 ,0
Exp/Cntr=0.3,0.1

Type RM Length L Ch R = 1 ,72694   ,530.7,527.9,515.7
XS GIS Cut Line= 3
2259043.21968497375006.7224900572258565.58907856375501.330096647
2258444.26123722375720.264041975
#Sta/Elev= 30
       0 2857.45      49 2852.55    75.7 2846.57   112.8 2833.53   184.7 2797.47
     204 2790.54   221.4 2788.19   258.8 2786.72   267.9 2782.92     277 2781.73
   307.7  2784.7   339.5 2784.78   367.8 2787.03   398.2 2785.78  409.63 2783.11
   418.4 2781.93  429.662783.331   450.3 2785.75   566.2 2787.44     610 2789.77
   632.8 2793.82   683.6 2810.96   713.8 2819.22   728.8 2820.85   757.2 2820.44
   794.3 2814.68     833 2811.42     862 2816.14   910.3 2835.84   937.9 2842.84
#Mann= 5 ,-1 , 0
       0      .1       0  406.53     .06       0  409.63    .045       0
  429.66     .06       0  564.93      .1       0
#XS Ineff= 2 , 0
          367.29 2789.25
Permanent Ineff=
       F       F
Bank Sta=409.63,429.66
XS Rating Curve= 0 ,0
Exp/Cntr=0.3,0.1

Type RM Length L Ch R = 1 ,72166   ,279,283.4,279.8
XS GIS Cut Line= 3
2258623.08076148374794.9168113172258498.08068338375031.027887642
2258204.40312114375640.851471141
#Sta/Elev= 30
       0 2836.04    19.7 2836.34    38.2 2834.74    60.9 2830.63    80.4 2825.25
   103.9 2816.49   119.9 2808.77   131.3 2801.81   160.7 2786.38   187.2 2775.78
     202 2775.29   231.3 2776.43     261 2775.66   273.72774.349   293.8    2772
   304.1 2772.53  312.942774.497   333.9 2777.48   366.7 2778.84   399.4 2778.45
   423.8 2777.19   457.7 2778.45   483.2 2777.33   499.4 2778.57   541.5 2779.19
     567 2781.89   585.2 2785.92   665.8 2789.17     800 2796.81     944 2806.88
#Mann= 7 ,-1 , 0
       0      .1       0    3.77     .12       0  208.14      .1       0
   273.7    .045       0  312.94      .1       0  427.44     .06       0
  563.48      .1       0
#XS Ineff= 2 , 0
          226.37 2778.53
Permanent Ineff=
       F       F
Bank Sta=273.7,312.94
XS Rating Curve= 0 ,0
Exp/Cntr=0.3,0.1

Type RM Length L Ch R = 1 ,71883   ,438.9,453.3,465.6
XS GIS Cut Line= 3
2258382.18065272374765.8515807242258276.62508956374988.073577225
2257969.68082155375460.296057984
#Sta/Elev= 30
       0  2815.3    18.3 2814.05    29.6 2812.55    44.1 2809.27    65.4 2801.62
    73.2 2797.77    80.5 2793.32    91.4  2788.4    98.6 2784.49   113.2  2778.5
   134.9 2772.84  154.482771.984   167.6 2769.82  186.972771.541   222.1 2773.69
   275.1 2772.98   304.4 2771.43   341.6 2773.35   361.4 2772.97   415.9 2774.84
   466.8  2775.1   484.7  2777.4   513.7 2782.96   541.6 2790.55   584.4 2805.73
   603.7  2811.4   655.4 2824.39   693.7 2832.53   757.4 2840.44   809.2 2845.86
#Mann= 6 ,-1 , 0
       0     .12       0  154.48    .045       0  186.97     .12       0
   211.8      .1       0  232.43     .06       0  383.85      .1       0
#XS Ineff= 2 , 0
                          224.67         2775.95
Permanent Ineff=
       F       F
Bank Sta=154.48,186.97
XS Rating Curve= 0 ,0
Exp/Cntr=0.3,0.1

Type RM Length L Ch R = 1 ,71430   ,242.9,247.5,249.9
XS GIS Cut Line= 2
2258355.79192597374770.0182390662257723.84732372 374738.07374914
#Sta/Elev= 30
       0 2812.18    30.7  2808.6    43.8 2805.08    70.1 2800.39   109.5 2789.17
   142.4 2778.19   158.8  2774.1   188.4 2770.92   234.4 2769.14   256.8 2765.11
   270.5 2763.15   273.8 2763.24  281.952765.435   293.5 2766.96   306.6 2767.21
   336.4 2769.58   346.1 2771.36   355.9 2772.17   369.1 2774.93   388.8  2781.4
   395.2 2784.55     415 2796.31   429.8 2803.01   457.8 2809.78   474.2 2814.64
   490.6 2818.08   517.4 2822.05   554.9 2826.13   586.2 2828.72   632.8  2830.3
#Mann= 5 ,-1 , 0
       0     .12       0  204.69     .06       0   256.8    .045       0
  281.95     .06       0  380.68      .1       0
Bank Sta=256.8,281.95
XS Rating Curve= 0 ,0
Exp/Cntr=0.3,0.1

Type RM Length L Ch R = 1 ,71182   ,281.9,286,287.3
XS GIS Cut Line= 2
2258439.12509264374607.5182359812257915.51426323374465.851524562
#Sta/Elev= 30
       0 2817.81    50.1 2807.56    77.3 2802.35    90.9 2800.31   105.2 2796.37
   192.9 2778.75   216.7 2773.17   226.9 2769.99   233.6 2768.56   250.6 2765.81
   265.7 2764.35     288 2762.94   318.6  2762.1   328.8 2761.14   333.32760.095
     339 2758.97   349.2 2758.28     356 2758.66  364.532760.034   400.2  2762.8
   410.2 2765.82   421.9 2770.82   430.8 2775.83   447.6 2786.64     458 2792.31
   485.3 2802.88   498.4 2806.16   512.3  2808.7   532.7 2810.93   542.4 2810.82
#Mann= 5 ,-1 , 0
       0     .12       0  299.48     .06       0   333.3    .045       0
  364.53     .06       0  425.59      .1       0
Bank Sta=333.3,364.53
XS Rating Curve= 0 ,0
Exp/Cntr=0.3,0.1

Type RM Length L Ch R = 1 ,70896   ,216.2,214.7,213.5
XS GIS Cut Line= 2
2258500.23619089374408.9070846442258036.34735489374179.740220144
#Sta/Elev= 30
       0 2818.65    67.2 2802.76    78.2 2800.59   103.8 2793.11   133.3 2785.24
     148 2780.16   173.3 2770.34   191.6  2762.7   206.3 2758.08   214.1 2756.65
   238.6  2754.6   264.8 2754.16   277.2 2752.06   286.8 2750.76   294.1 2750.34
  313.922752.274   334.1 2756.17   352.7 2757.55   358.6  2758.8   367.3 2761.95
   374.6 2765.31   378.2 2767.58   389.2 2772.11   411.2 2778.37     437 2783.75
   447.8 2785.47   455.1  2787.5   462.4 2788.45   505.6 2796.29   517.4 2797.82
#Mann= 4 ,-1 , 0
       0     .12       0   277.2    .045       0  313.92     .06       0
  458.79      .1       0
Bank Sta=277.2,313.92
XS Rating Curve= 0 ,0
Exp/Cntr=0.3,0.1

Type RM Length L Ch R = 1 ,70681   ,126.1,116.5,103.4
XS GIS Cut Line= 3
2258612.41425513374175.362868851 2258304.1200447374092.083393825
2258074.30072419374176.163633034
#Sta/Elev= 30
       0 2831.93    22.3 2827.27    42.7 2822.25    73.3 2815.06   117.5 2798.53
     148 2784.43   158.2 2781.21   185.8    2774   219.4 2760.84   229.6 2756.06
   236.4 2751.79   240.7 2749.76   246.6  2748.2   266.82748.434   279.4 2748.93
   294.2 2748.04   307.8 2749.04   321.4 2748.89   342.4 2750.11     372 2750.38
   380.8 2750.54   391.3 2752.13   438.9 2761.21   478.6 2767.16   489.1 2769.76
   506.4 2772.89     524 2777.31     531  2778.3     552 2785.17   564.1 2788.52
#Mann= 7 ,-1 , 0
       0      .1       0    42.7     .12       0   185.8     .06       0
   240.7    .045       0   266.8     .06       0   321.4     .12       0
     372     .06       0
Bank Sta=240.7,266.8
XS Rating Curve= 0 ,0
Exp/Cntr(USF)=0,0
Exp/Cntr=0.3,0.1

Type RM Length L Ch R = 1 ,70565   ,234.6,234.5,230.1
XS GIS Cut Line= 3
2258571.06971064373829.7402639842258186.34738298374125.573661804
2258054.40309305374168.629349977
#Sta/Elev= 30
       0 2805.14    37.1 2798.54    61.9 2792.82    90.9  2785.1   107.4 2779.04
   142.5 2773.67   153.3 2770.66   180.2 2768.12   190.5 2766.01   202.2 2762.52
   213.9  2757.2   235.7 2749.72   248.2 2748.33   277.1 2747.19   281.8 2746.66
  288.562744.757   293.2 2743.34     302 2742.71  313.132745.136   323.9 2745.54
   361.3 2744.67   370.7 2745.92   380.6  2748.1   413.7 2748.83   430.3 2750.48
   473.6  2759.4   519.2 2766.56   560.2 2774.77   604.9 2787.82   624.1 2792.75
#Mann= 6 ,-1 , 0
       0      .1       0  108.47     .12       0  288.56    .045       0
  313.13     .12       0  373.36     .06       0  576.44      .1       0
#XS Ineff= 2 , 0
                          356.93         2748.44
Permanent Ineff=
       F       F
Bank Sta=288.56,313.13
XS Rating Curve= 0 ,0
Exp/Cntr=0.3,0.1

Type RM Length L Ch R = 1 ,70330   ,184.2,187.3,188.9
XS GIS Cut Line= 2
2258396.85274568373603.5406308132257943.03448983374158.826850501
#Sta/Elev= 30
       0 2780.51    19.3  2772.5    39.9 2766.66    86.6 2757.11   128.9    2747
   142.9 2744.54   162.8  2742.1   188.2 2740.72   213.7 2740.38   248.1 2741.57
   268.9 2741.22   284.4    2740   311.1 2738.43   331.1 2738.88   350.12738.559
   366.7 2738.33   383.2 2739.53   408.6 2738.94     425 2737.96   429.8 2738.98
   442.5 2744.45   459.4 2753.08   486.6 2765.27     502 2770.08   514.5 2775.11
     554 2786.78   595.2 2793.74   626.6 2796.76   657.7 2799.52   717.1 2802.25
#Mann= 6 ,-1 , 0
       0      .1       0   142.9     .12       0   284.4     .06       0
   331.1    .045       0   350.1     .06       0   408.6      .1       0
Bank Sta=331.1,350.1
XS Rating Curve= 0 ,0
Exp/Cntr(USF)=0,0
Exp/Cntr=0.3,0.1

Type RM Length L Ch R = 1 ,70143   ,466.9,468.9,459.3
XS GIS Cut Line= 2
2258337.06591356373503.0831088872257647.48231897374125.999842063
#Sta/Elev= 30
       0 2783.01    29.3 2779.39    63.9  2772.6   101.5 2760.59   132.4 2748.02
   147.1 2743.68   166.4  2740.2   238.5 2736.68   275.7  2737.5   352.6 2733.84
     383  2734.9   403.4 2732.76   418.4 2732.82  425.372731.466   430.9 2730.04
   440.5 2729.47   445.3 2729.88  448.282731.333   465.2 2743.17   484.7 2751.59
     498 2756.16   547.5 2768.79   596.2 2775.06   614.8 2776.35   661.6 2775.44
   710.2 2775.65   726.3  2774.8   784.4 2775.02   909.8  2777.9   929.3 2777.46
#Mann= 7 ,-1 , 0
       0      .1       0  159.84     .12       0  317.68     .06       0
  425.37    .045       0  448.28     .06       0   473.6     .12       0
   527.9      .1       0
#XS Ineff= 2 , 0
          380.31  2737.5
Permanent Ineff=
       F       F
Bank Sta=425.37,448.28
XS Rating Curve= 0 ,0
Exp/Cntr=0.3,0.1

Type RM Length L Ch R = 1 ,69674   ,447.8,471,473.9
XS GIS Cut Line= 3
2257947.48237513373242.6666349772257699.56587622373540.583361983
2257359.98256588373850.999735892
#Sta/Elev= 30
       0 2782.51    68.3 2776.26    91.4 2772.43   140.6 2759.93   159.7 2756.27
   193.9 2744.56   225.1 2732.05   240.8 2727.57   257.9 2726.43   275.6 2723.46
  293.132722.269   312.9 2720.92   325.72722.412     338 2723.73   373.9 2722.34
   414.9 2722.07   451.3 2723.75   473.4 2721.81     485 2722.17   521.9 2728.15
   547.7 2738.88   570.9 2750.47   580.2 2754.09   589.1 2759.28   602.4  2765.5
   624.6 2771.92   642.4 2775.38   669.1 2778.01   707.9 2780.08   847.7 2785.44
#Mann= 7 ,-1 , 0
       0     .12       0   235.3     .06       0  293.13    .045       0
   325.7     .06       0  383.71      .1       0  610.93     .12       0
  674.62      .1       0
Bank Sta=293.13,325.7
XS Rating Curve= 0 ,0
Exp/Cntr=0.3,0.1

Type RM Length L Ch R = 1 ,69203   ,234,239.2,242.8
XS GIS Cut Line= 2
 2257932.1700698373165.062459484 2257154.3920978373291.798426479
#Sta/Elev= 30
       0 2782.85    20.7 2780.17   103.8 2771.91     137 2767.22   216.8 2749.42
   236.8 2743.53   289.6 2725.94   313.2 2719.38   323.2  2717.8   358.2 2716.12
   376.4 2713.49   399.6 2714.24   406.3 2713.72  408.732712.873   412.9 2711.69
   426.2 2710.32  441.432712.385   456.1  2715.4     496 2717.97   522.6 2720.69
   539.3 2727.48   545.9 2732.15   565.8 2743.27   586.8 2750.47   599.1 2754.03
   612.5 2757.15   665.6 2765.21   715.4 2775.69   745.3 2780.61     788 2786.28
#Mann= 5 ,-1 , 0
       0     .12       0  350.12     .06       0  408.73    .045       0
  441.43     .06       0   478.6      .1       0
Bank Sta=408.73,441.43
XS Rating Curve= 0 ,0
Exp/Cntr=0.3,0.1

Type RM Length L Ch R = 1 ,68964   ,196.5,204.6,209.6
XS GIS Cut Line= 3
2257921.75342397372987.9791522322257459.94758905 373003.60412097
2257003.35040514 373014.02076681
#Sta/Elev= 30
       0 2784.65    82.2 2776.36   115.1 2772.22     207 2758.32   220.1 2754.13
     230 2752.32   275.9 2739.79   321.9 2719.52   341.6 2714.41   356.8 2712.02
  365.382708.257   367.8 2707.03  376.87 2708.16   390.7 2710.18   413.8 2710.24
     486 2707.44   528.7 2708.16   538.5 2710.44   584.4 2716.71   600.9  2719.9
   653.2 2737.07   659.9 2738.44   692.7 2750.98   709.2 2755.62   725.6 2758.82
   768.2 2773.57   791.2 2779.06   804.3 2780.95   824.8 2781.88   918.8 2779.11
#Mann= 6 ,-1 , 0
       0      .1       0   31.76     .12       0  365.38    .045       0
  376.87     .12       0   419.9     .06       0  534.24      .1       0
Bank Sta=365.38,376.87
XS Rating Curve= 0 ,0
Exp/Cntr=0.3,0.1

Type RM Length L Ch R = 1 ,68759   ,339.5,350.8,347.9
XS GIS Cut Line= 2
2257994.66994481372805.6875220542256973.83668464372843.881671399
#Sta/Elev= 30
       0 2780.63    63.3 2775.04   171.6 2763.48   213.7 2757.74   258.1 2752.99
   299.7 2746.97   316.1 2744.31   371.9 2731.25   417.9 2716.18   434.3 2710.12
   483.2 2707.43  514.052703.996   532.8    2702  550.062703.941   562.3 2705.24
     605  2705.6   614.8 2703.01   618.1 2702.75     628 2703.93   634.5 2705.56
   661.1 2707.04   670.8  2708.4   687.1 2713.02   727.5 2732.72   798.7 2760.67
   818.4 2766.92   831.5 2770.09   874.2  2774.6     976 2783.17  1021.5 2785.61
#Mann= 6 ,-1 , 0
       0      .1       0  122.71     .12       0  511.49     .06       0
  514.05    .045       0  550.06     .06       0  659.04      .1       0
Bank Sta=514.05,550.06
XS Rating Curve= 0 ,0
Exp/Cntr=0.3,0.1

Type RM Length L Ch R = 1 ,68409   ,292.6,295.2,294.6
XS GIS Cut Line= 4
2257909.92470747372730.1502715652257625.20250788372653.761316732
 2257274.5079993372542.6503184742256996.73001155372506.192058057
#Sta/Elev= 30
       0 2755.24    49.1 2749.16   120.4  2738.8   212.1 2727.21   263.1 2717.06
     315 2708.14     338 2705.73   383.4 2703.02   451.9 2702.26   472.6 2702.83
   527.6 2701.56   541.4 2699.81   565.5 2700.38   582.7 2699.26  597.562699.285
   618.2 2696.85  626.712698.812   658.4  2708.4   681.8  2718.9   701.6 2729.33
   711.5 2735.35   721.5 2737.81   728.1 2741.93   744.6 2747.91   759.1  2751.8
   777.7 2755.06   810.8 2757.88   840.6 2758.57   900.1 2761.79   942.8 2761.13
#Mann= 7 ,-1 , 0
       0      .1       0   48.87     .12       0   395.9     .06       0
  547.16      .1       0  597.56    .045       0  626.71      .1       0
  693.27      .1       0
Bank Sta=597.56,626.71
XS Rating Curve= 0 ,0
Exp/Cntr=0.3,0.1

Type RM Length L Ch R = 1 ,68113   ,290.3,280.7,275
XS GIS Cut Line= 3
2257975.89668839 372476.678009482257724.16064331372405.497705638
2257151.24413823 372205.84488973
#Sta/Elev= 30
       0 2772.24    46.2 2769.61    90.5 2765.14   155.9 2753.42   230.4 2735.39
   254.2 2726.04   274.9 2716.59   323.5 2703.15   367.8 2699.66   395.3 2698.86
   431.2 2694.23   448.6 2694.51   469.5 2698.53   483.8  2699.1   518.1  2697.4
     532 2695.95   538.9 2693.95   574.7 2695.21     5832693.943     598 2692.53
   609.22694.215   643.2 2695.02   667.5 2707.83   691.8  2723.4   702.2 2728.68
   738.4  2741.8   785.6 2755.46   798.1 2757.75   827.3 2760.98   868.3 2761.87
#Mann= 6 ,-1 , 0
       0      .1       0   58.68     .12       0   471.6     .06       0
  560.02      .1       0     583    .045       0   609.2      .1       0
#XS Ineff= 2 , 0
          476.51 2707.01
Permanent Ineff=
       F       F
Bank Sta=583,609.2
XS Rating Curve= 0 ,0
Exp/Cntr=0.3,0.1

Type RM Length L Ch R = 1 ,67833   ,507.9,493.5,481
XS GIS Cut Line= 2
2258036.66067447371987.0946710562257126.93841255372115.566855058
#Sta/Elev= 30
       0 2770.71    53.3 2768.47   106.3 2764.08   235.5 2748.71   268.6  2743.4
   305.1 2735.88   334.5 2727.34   378.2 2709.59   401.2 2702.46   417.7 2699.02
   464.1 2696.11   474.1 2694.24     484 2689.51  490.442689.394  522.332689.876
   570.1 2691.77   583.4 2687.51   586.7 2687.46   609.9 2692.64   653.8  2690.8
   699.4 2692.28   709.3 2691.76   719.2 2692.84   732.5 2697.62   742.4 2702.33
   802.3 2737.46   825.1 2746.91   838.5 2750.41   855.1 2752.55   918.7 2754.78
#Mann= 7 ,-1 , 0
       0      .1       0  236.56     .12       0   443.7      .1       0
  490.44    .045       0  522.33      .1       0  539.64     .06       0
  712.71      .1       0
#XS Ineff= 2 , 0
                          692.13         2696.21
Permanent Ineff=
       F       F
Bank Sta=490.44,522.33
XS Rating Curve= 0 ,0
Exp/Cntr=0.3,0.1

Type RM Length L Ch R = 1 ,67339   ,400.7,403.6,402.6
XS GIS Cut Line= 2
2257345.68863122371450.6364263892257059.23021464 372092.99767448
#Sta/Elev= 30
       0  2748.8    27.4  2748.8      49 2747.62    84.9 2742.63    92.1 2740.04
    99.3 2739.21   113.6 2734.44   142.4 2726.88   163.9 2720.02   185.5 2710.64
   196.3 2706.96   217.8  2696.3   235.8 2690.61   296.8 2685.72   314.8 2686.14
     340 2684.54     358 2685.63   383.1 2685.61     4042683.828   411.8 2682.06
  425.272684.196   436.9 2686.67   454.9 2688.68   480.1 2696.46   494.6 2702.22
   548.3 2716.65   555.5 2717.66   586.6 2725.75   634.5 2736.21   703.3 2749.98
#Mann= 6 ,-1 , 0
       0      .1       0  150.98     .12       0  345.94      .1       0
     404    .045       0  425.27     .06       0  572.82      .1       0
Bank Sta=404,425.27
XS Rating Curve= 0 ,0
Exp/Cntr=0.3,0.1

Type RM Length L Ch R = 1 ,66936   ,313.6,316.8,318.5
XS GIS Cut Line= 2
2256942.91056539371436.7476746442256748.46640047372091.261457473
#Sta/Elev= 30
       0 2739.21    30.3 2738.72    57.7 2736.85      92 2732.62   105.6 2728.53
   119.3  2722.9   126.2 2721.34   139.9 2714.75   153.6  2709.2   167.3 2704.86
     181 2699.26   191.2  2694.2   204.9 2689.45   215.2 2686.99   263.1 2683.91
   331.5 2683.62   362.3 2680.88   375.72680.599   396.6 2679.05   406.8 2679.89
  411.632681.236   420.5  2683.4   454.7 2685.54   475.3 2688.38   492.4 2692.23
   533.5 2704.03   547.2 2706.66   601.9 2719.93   656.7 2731.21   682.8 2734.65
#Mann= 6 ,-1 , 0
       0      .1       0   67.43     .12       0  352.95     .06       0
   375.7    .045       0  411.63     .06       0  483.31      .1       0
#XS Ineff= 2 , 0
          327.62 2688.64
Permanent Ineff=
       F       F
Bank Sta=375.7,411.63
XS Rating Curve= 0 ,0
Exp/Cntr=0.3,0.1

Type RM Length L Ch R = 1 ,66619   ,294.1,306,317
XS GIS Cut Line= 2
2256727.63278072371388.1365513952256352.63287455372063.483625889
#Sta/Elev= 30
       0 2719.98   100.1 2714.47   107.6 2713.18   144.2 2709.48   175.2 2704.83
   224.5 2699.08   246.5 2695.59     269 2690.62   293.8  2684.2   310.3 2681.61
   329.1  2680.8   347.8 2678.01   366.2 2679.81   377.8 2680.04  396.062678.757
   400.4  2677.2   404.1 2676.88   411.6 2676.95  422.24 2678.59   437.9 2681.12
   445.4 2683.07   471.7 2686.89   494.2 2693.13   501.7 2694.49   527.9 2703.23
   554.7 2710.15   591.7 2714.98     633  2718.7   726.8 2725.13   772.5 2727.55
#Mann= 4 ,-1 , 0
       0     .12       0  396.06    .045       0  422.24     .06       0
   518.4      .1       0
Bank Sta=396.06,422.24
XS Rating Curve= 0 ,0
Exp/Cntr=0.3,0.1

Type RM Length L Ch R = 1 ,66313   ,193,190.1,184.8
XS GIS Cut Line= 3
2256706.79948905371384.6641173962256267.56349088371533.969921142
2255958.53556564371657.233782232
#Sta/Elev= 30
       0 2717.28    33.7 2713.05   148.1 2702.05   200.4 2694.76   224.3 2690.74
   278.2 2684.25   307.5 2677.86   323.6 2678.09   331.7  2676.5  362.642675.671
   373.3 2673.23   376.8 2673.07  401.84 2675.27     408 2675.78   421.8 2678.45
   439.1 2678.53   456.4 2680.34     466 2682.77   499.5 2694.26   523.4 2700.67
   565.8 2707.03   577.8 2707.23   590.6 2708.86   615.6 2710.62     652 2712.68
   661.2 2712.57   679.1 2713.88     704 2714.62   728.3 2716.48   796.6 2717.97
#Mann= 6 ,-1 , 0
       0     .12       0  253.08     .06       0  362.64    .045       0
  401.84     .06       0  493.59      .1       0  744.36     .12       0
Bank Sta=362.64,401.84
XS Rating Curve= 0 ,0
Exp/Cntr=0.3,0.1

Type RM Length L Ch R = 1 ,66123   ,432.7,445.6,441.2
XS GIS Cut Line= 3
2256643.61687264371172.8761551382256379.03341231371270.792625979
2255948.82495514371533.292757139
#Sta/Elev= 30
       0 2703.35    96.4 2694.47   159.1 2689.52     271 2683.99   327.6 2680.27
   337.7 2678.45   347.9  2675.3   354.2  2674.2     366  2675.3   398.3 2675.83
   403.22675.167   412.1 2672.87   430.8 2673.13   439.22675.034   449.9 2676.28
     469 2675.78   488.1  2676.1   499.1 2678.43   505.4 2680.72     518 2681.85
   524.3 2684.25     531 2685.43   562.1 2689.31   569.7 2690.95   588.3 2693.44
   656.6 2701.06   696.5 2704.29   712.4 2704.76   724.4  2705.8   786.1 2707.49
#Mann= 7 ,-1 , 0
       0     .12       0  315.13     .06       0   403.2    .045       0
   439.2     .06       0  508.78     .12       0  616.04      .1       0
  646.05     .12       0
Bank Sta=403.2,439.2
XS Rating Curve= 0 ,0
Exp/Cntr=0.3,0.1

Type RM Length L Ch R = 1 ,65677   ,296.3,294.3,292.4
XS GIS Cut Line= 3
2256600.90829664371044.2996406412256309.24155714371021.730131984
2255788.40828122 371096.38286981
#Sta/Elev= 30
       0 2692.35    37.7 2686.79    80.5 2682.39   139.7 2679.22   274.6 2675.57
   317.6 2672.09   347.4 2672.19   373.9 2670.49   387.2 2670.93   403.8 2670.53
   463.5 2672.41     480 2671.39   503.9 2671.96   523.1 2670.53   559.5 2671.51
   566.2 2670.38   573.5 2670.23   592.7 2668.21   599.3 2669.14     6032670.341
   647.8 2684.84   655.6 2686.97   665.6 2688.62   685.5 2690.77   718.9 2693.48
   735.2 2695.78   758.4 2696.48   771.6 2697.56   785.1 2697.39   818.7 2698.23
#Mann= 5 ,-1 , 0
       0     .12       0  414.73     .06       0   573.5    .045       0
     603     .06       0  817.61      .1       0
#XS Ineff= 2 , 0
          461.23 2673.97
Permanent Ineff=
       F       F
Bank Sta=573.5,603
XS Rating Curve= 0 ,0
Exp/Cntr=0.3,0.1

Type RM Length L Ch R = 1 ,65383   ,392.9,370.6,372.2
XS GIS Cut Line= 2
2256644.31109697370806.4523473082256014.10271172 370818.60521014
#Sta/Elev= 30
       0 2689.62    59.2 2684.51      81 2681.64   113.8 2679.06   130.2  2678.4
   186.4 2674.92     209 2673.11   223.2 2671.09   238.5 2669.73   248.4  2669.5
   261.5 2669.85     291 2668.62   304.1 2669.12   330.5 2669.25   346.6 2669.95
   383.8 2668.47   445.2 2668.19   480.8 2669.22  483.36 2668.88   491.2 2667.31
   497.6 2666.85   517.6 2666.95  529.082668.021     547 2668.25   551.1 2668.77
   554.4  2669.7   576.5 2678.68   589.6 2681.61   612.6 2683.56   630.3 2683.04
#Mann= 4 ,-1 , 0
       0     .12       0  483.36    .045       0  529.08     .12       0
  542.07     .06       0
Bank Sta=483.36,529.08
XS Rating Curve= 0 ,0
Exp/Cntr=0.3,0.1

Type RM Length L Ch R = 1 ,65012   ,545.7,449.7,579.7
XS GIS Cut Line= 3
2256791.88068372370440.1328699742256059.24172905370487.008104309
2255371.74179173370834.230178893
#Sta/Elev= 30
       0 2697.28    47.3 2696.75    87.4 2694.69   146.8 2693.85   170.9 2692.38
   229.6 2685.11   284.9 2674.89     397  2668.8  471.95 2667.12   557.8 2666.91
  560.432666.965   580.8 2667.54   603.8 2666.91     699 2667.12   705.7 2668.09
   720.1 2673.31   735.4 2674.76   787.1 2670.19   801.6 2669.63   900.8 2670.51
  1047.9 2673.13  1136.4 2675.95  1191.2 2679.38  1224.3 2679.63  1272.1 2681.54
  1294.1 2681.38  1371.3 2683.57  1404.4 2684.95    1428 2687.33  1504.3 2688.12
#Mann= 9 ,-1 , 0
       0      .1       0  234.46     .12       0  468.95    .045       0
  471.95    .045       0  560.43     .12       0  800.81     .06       0
  910.66      .1       0 1108.66     .06       0 1232.36      .1       0
Bank Sta=471.95,560.43
XS Rating Curve= 0 ,0
Exp/Cntr=0.3,0.1

Type RM Length L Ch R = 1 ,64562   ,489.2,453.4,440.3
XS GIS Cut Line= 2
2256845.70012988 369884.577550652255493.26943581370179.716396064
#Sta/Elev= 30
       0 2701.02    27.7 2695.88    47.2 2693.98    55.2 2692.72     101 2689.12
   114.4    2687   171.5  2680.1     242  2673.3   282.3 2670.88   292.5 2669.68
   322.7 2667.65   342.7 2667.92   350.2 2666.98  1077.9 2666.87  1080.7 2666.88
  1088.2 2667.38    1105 2667.15  1131.9 2667.88  1153.6 2669.38    1169 2671.88
    1189 2672.67  1215.7 2677.01  1242.7 2682.24  1252.8 2684.96    1283 2695.09
  1303.9 2699.12  1323.2 2701.89  1346.8 2704.22    1367 2704.75  1384.3 2703.55
#Mann= 7 ,-1 , 0
       0      .1       0  197.52     .12       0  328.56    .025       0
   350.2    .045       0  1080.7      .1       0 1092.75     .06       0
 1208.41      .1       0
Bank Sta=350.2,1080.7
XS Rating Curve= 0 ,0
Exp/Cntr=0.3,0.1

Type RM Length L Ch R = 1 ,64109   ,838.8,689.6,523.6
XS GIS Cut Line= 3
2256781.98261643369376.4051934292255483.79221902369757.870040504
2254891.19972331370581.783058949
#Sta/Elev= 30
       0 2708.15    50.1 2703.16   117.6  2693.8   167.8 2682.36   210.1    2676
   241.6 2673.26   310.6 2670.88   333.9 2668.99   340.7 2667.03   344.2 2666.91
  1259.4 2667.07  1267.3 2668.55  1281.1 2674.48  1305.1 2681.36  1322.2 2682.94
  1371.6 2684.31  1468.6 2684.86  1541.4 2679.44  1626.2 2685.26    1703 2688.59
  1836.1 2691.92  1884.9 2691.01  2006.1 2683.55  2054.9 2685.17  2078.9 2688.66
  2111.3 2689.66  2195.7 2687.22  2232.4 2688.16  2311.1 2687.13    2368 2688.85
#Mann= 9 ,-1 , 0
       0      .1       0   59.71      .1       0  159.83    .025       0
   340.7    .045       0  1259.4     .06       0  1315.5      .1       0
 1361.31     .06       0 1776.08     .12       0 1823.02     .06       0
Bank Sta=340.7,1259.4
XS Rating Curve= 0 ,0
Exp/Cntr=0.3,0.1

Type RM Length L Ch R = 1 ,63420   ,778.6,722.7,719.2
XS GIS Cut Line= 3
2256465.74478528368493.7834614122255127.99162306369402.980088636
2254528.36699574370177.294027435
#Sta/Elev= 30
       0 2689.38    48.6 2684.55    60.5 2684.33    88.3 2681.69   132.6 2681.88
     243  2674.7   255.4 2674.02   322.3 2667.07   326.3 2666.91  1429.2    2667
  1429.3 2667.01  1459.9 2669.24  1618.1 2672.56  1679.1 2671.34  1778.3 2673.23
  1790.8 2672.81  1865.5 2673.59    1907 2673.35    1936 2671.51  2064.6  2677.1
  2111.5 2678.38  2123.9 2679.39  2151.3 2678.94  2312.7 2682.05  2429.6 2682.73
  2487.9 2684.58  2551.2 2683.62  2562.6 2682.81  2590.1 2683.28  2596.8  2682.6
#Mann= 7 ,-1 , 0
       0     .12       0     243    .025       0   322.3    .045       0
  1429.2    .045       0  1429.3     .06       0 2230.19     .12       0
 2313.69     .06       0
Bank Sta=322.3,1429.2
XS Rating Curve= 0 ,0
Exp/Cntr=0.3,0.1
